--- DRYRN.prj (project) ---

Proj Title=DRYRN
Current Plan=p01
Default Exp/Contr=0,0
English Units
Geom File=g01
Flow File=f01
Plan File=p01
BEGIN DESCRIPTION:
----------MODEL BY WOOD PLC 2022----------
AFH study
Randolph County, WV
HEC-RAS Version: RAS 6.2
Vertical Datum: NAVD88
Projection: NAD 1983 StatePlane West Virginia S FIPS 4702 (US Feet)
Terrain: 1-meter LIDAR (FEMA Region III 3DEP collected 2016-2018)
Land Use: 2019 NLCD
Hydrologic Method:
WV SIR2010-5033 regression equations
Additional Model Notes:
None
END DESCRIPTION:
DSS File=dss
DSS Export Rating Curves= 0
DSS Export Rating Curve Sorted= 0
DSS Export Volume Flow Curves= 0
DXF OffsetX= 0
DXF OffsetY= 0
DXF ScaleX= 0
DXF ScaleY= 0

--- DRYRN.p01 (plan) ---

Plan Title=Floodplain
Program Version=6.20
Short Identifier=Floodplain
Geom File=g01
Flow File=f01
Subcritical Flow
K Sum by GR= 0
Std Step Tol= 0.01
Critical Tol= 0.01
Num of Std Step Trials= 20
Max Error Tol= 0.3
Flow Tol Ratio= 0.001
Split Flow NTrial= 30
Split Flow Tol= 0.02
Split Flow Ratio= 0.02
Log Output Level= 0
Friction Slope Method= 1
Unsteady Friction Slope Method= 2
Unsteady Bridges Friction Slope Method= 1
Parabolic Critical Depth
Global Vel Dist= 0 , 0 , 0
Global Log Level= 0
CheckData=True
Encroach Param=-1 ,0,0, 0
Computation Interval=0.1SEC
Output Interval=1SEC
Instantaneous Interval=Max Profile
Mapping Interval=1HOUR
Computation Time Step Use Courant=        0
Computation Time Step Use Time Series=    0
Computation Time Step Count To Double=0
Computation Time Step Max Doubling=0
Computation Time Step Max Halving=0
Computation Time Step Residence Courant=0
Run HTab= 0
Run UNet= 0
Run Sediment= 0
Run PostProcess= 0
Run WQNet= 0
Run RASMapper=-1
UNET Theta= 0
UNET Theta Warmup= 0
UNET ZTol= 0
UNET ZSATol= 0
UNET MxIter= 0
UNET Max Iter WO Improvement= 0
UNET MaxInSteps= 0
UNET DtIC= 0
UNET DtMin= 0
UNET MaxCRTS= 0
UNET WFStab= 0
UNET SFStab= 0
UNET WFX= 1
UNET SFX= 1
UNET Gravity=32.174
UNET 1D Methodology=Finite Difference
UNET DSS MLevel= 1
UNET Pardiso=0
UNET DZMax Abort= 0
UNET Use Existing IB Tables= 0
UNET Froude Reduction=False
UNET Froude Limit= 0
UNET Froude Power= 0
UNET D1 Cores= 0
UNET WindReference=Eulerian
UNET WindDragFormulation=Hsu (1988)
UNET D2 Coriolis=0
UNET D2 Cores= 0
UNET D2 Theta= 1
UNET D2 Theta Warmup= 1
UNET D2 Z Tol= 0.01
UNET D2 Volume Tol= 0.01
UNET D2 Max Iterations= 20
UNET D2 Equation= 0
UNET D2 RampUpFraction=0.1
UNET D2 TimeSlices= 1
UNET D2 Turbulence Formulation=Non-Conservative (original)
UNET D2 Eddy Viscosity=0.3
UNET D2 Transverse Eddy Viscosity=0.1
UNET D2 Smagorinsky Mixing=0
UNET D2 BCVolumeCheck=0
UNET D2 Cores=0
UNET D2 SolverType=PARDISO (Direct)
UNET D2 Minimum Iterations= 2147483647
UNET D2 Maximum Iterations= 2147483647
UNET D2 Restart Number= 10
UNET D2 Relaxation Coeff=1.3
UNET D2 SOR Precondition Iterations= 10
UNET D2 ILUT Maximum Fill= 8
UNET D2 ILUT Tolerance=1E-08
UNET D1D2 MaxIter= 0
UNET D1D2 ZTol=0.01
UNET D1D2 QTol=0.1
UNET D1D2 MinQTol=1
DSS File=dss
Write IC File= 0
Write IC File at Fixed DateTime=0
Write IC File at Sim End=0
Echo Input=False
Echo Parameters=False
Echo Output=False
Write Detailed= 0
HDF Write Warmup=0
HDF Write Time Slices=0
HDF Flush=0
HDF Compression= 1
HDF Chunk Size= 1
HDF Spatial Parts= 1
HDF Use Max Rows=0
HDF Fixed Rows= 1
Calibration Method= 0
Calibration Iterations= 20
Calibration Max Change=0.05
Calibration Tolerance=0.2
Calibration Maximum=1.5
Calibration Minimum=0.5
Calibration Optimization Method= 1
WQ AD Non Conservative
WQ ULTIMATE=-1
WQ Max Comp Step=1HOUR
WQ Output Interval=15MIN
WQ Output Selected Increments= 0
WQ Output face flow=0
WQ Output face velocity=0
WQ Output face area=0
WQ Output face dispersion=0
WQ Output cell volume=0
WQ Output cell surface area=0
WQ Output cell continuity=0
WQ Output cumulative cell continuity=0
WQ Output face conc=0
WQ Output face dconc_dx=0
WQ Output face courant=0
WQ Output face peclet=0
WQ Output face adv mass=0
WQ Output face disp mass=0
WQ Output cell mass=0
WQ Output cell source sink temp=0
WQ Output nsm pathways=0
WQ Output nsm derived pathways=0
WQ Create Restart=0
WQ Fixed Restart=0
WQ System Summary=0
WQ Write To DSS=0
Sorting and Armoring Iterations= 10
XS Update Threshold= 0.02
Bed Roughness Predictor= 0
Hydraulics Update Threshold= 0.02
Energy Slope Method= 1
Volume Change Method= 1
Sediment Retention Method= 0
Sediment TS Multiplier= 1
Warm Up Method= 0
XS Weighting Method= 0
Number of US Weighted Cross Sections= 1
Number of DS Weighted Cross Sections= 1
Upstream XS Weight=0
Main XS Weight=1
Downstream XS Weight=0
Number of DS XS's Weighted with US Boundary= 1
Upstream Boundary Weight= 1
Weight of XSs Associated with US Boundary= 0
Number of US XS's Weighted with DS Boundary= 1
Downstream Boundary Weight= 0.5
Weight of XSs Associated with DS Boundary= 0.5
Percentile Method= 0
Sediment Output Level= 3
Mass or Volume Output= 0
Output Increment Type= 1
Profile and TS Output Increment= 1
Transport Output Increment 1
XS Output Flag= 0
XS Output Increment= 10
Read HDF5 Sediment Hotstart= 0
Sediment Hotstart Type= 0
Write Gradation File= 0
Read Gradation Hotstart= 0
Write HDF5 File= 1
Write Binary Output= 1
Write DSS Sediment File= 0
DSS Sediment Output Type= 1
SV Curve= 0
Specific Gage Flag= 0
Subcell Erosion Methods= 0
Subcell Deposition Methods= 0
Advection Scheme= 1
Matrix Solver= 0
Implicit Weighting Factor= 1
Maximum Outer Loop Convergence Iterations= 5
Convergence Maximum Absolute= 0.001
Convergence RMSE= 0.0001
Grain Fractions Max Abs Error= 0.001
Max Subgrid Regions= 1
Max Subgrid Length Scale= 3.402823E+38
Initial Layer Thickness= 3.402823E+38
Min Layer Thickness= 3.402823E+38
Max Layer Thickness= 3.402823E+38
Number of Layers= 5

--- DRYRN.f01 (steady flow) ---

Flow Title=Flow
Program Version=6.20
Number of Profiles= 1
Profile Names=P100yr
River Rch & RM=DRYRN,Main,14030
     403
River Rch & RM=DRYRN,Main,7727
     596
River Rch & RM=DRYRN,Main,3011
     673
Boundary for River Rch & Prof#=DRYRN,Main            , 1
Up Type= 0
Dn Type= 3
Dn Slope=0.00942
DSS Import GetInterval= 0
DSS Import GetPeak= 0
DSS Import FillOption= 0

--- DRYRN.g01 (geometry) ---

Geom Title=Geometry
Program Version=6.20

River Reach=DRYRN           ,Main
Reach XY= 30
     2274835.423      626203.535     2274436.767      626315.706
     2274284.468      626466.903     2274169.017      626436.087
     2273711.233      626781.313     2273550.434        626698.5
     2273361.169      626840.486     2273208.629      626781.833
     2272723.212      627108.917     2272277.379      628052.667
     2272097.171      628084.438     2272132.587      628355.792
2271938.59612137628623.058169917     2271694.045      628721.417
     2271528.941      629221.938     2271105.568      629585.737
2271210.97823466629986.123767501     2270631.456      630733.561
     2270377.067      630918.4572270336.93409628631251.144144425
     2269984.045      631648.669     2269757.881      631667.664
      2269379.77      631974.993     2269106.141      632687.675
     2268845.815      633023.297     2268054.422      633329.507
     2267323.524      633398.328     2267046.089      633312.146
     2266108.285      633594.784     2265835.173      634020.023

Type RM Length L Ch R = 1 ,14030   ,244.2,246.3,247.4
XS GIS Cut Line= 4
2274748.27525655626031.8837576962274817.63324147626178.367437203
 2274871.5759744626273.1242926152274912.92699685626501.490559722
#Sta/Elev= 30
       0 2340.54    14.7 2331.13    42.9 2311.95    54.5 2305.62    63.4 2302.71
    67.8  2301.8    85.5 2300.72   120.9 2301.44   129.8 2300.94   142.1  2301.6
   160.8  2301.3   179.1 2299.41   183.22298.425   189.5 2297.38   197.5 2297.18
   209.52298.391   211.3 2298.56   215.9 2300.46   225.1 2308.86   233.5 2314.31
   259.9 2323.77   291.5 2336.79     313 2346.36     335 2356.92   360.6 2371.11
   364.7 2372.67   397.2 2391.05   431.6 2407.01   454.1 2416.19   503.2  2430.9
#Mann= 3 ,-1,0
       0      .1       0   183.2    .045       0   209.5      .1       0
Bank Sta=183.2,209.5
XS Rating Curve= 0 ,0
Exp/Cntr=0.3,0.1

Type RM Length L Ch R = 1 ,13783   ,283.7,283.2,281.8
XS GIS Cut Line= 3
2274587.23144834626043.4036764832274572.73245259626213.318161224
2274688.55958729 626436.99355425
#Sta/Elev= 30
       0 2327.15    25.9    2316    45.9 2306.53      58 2301.78      70 2298.42
    94.1 2296.58   106.2 2296.55   134.3 2295.23   154.3 2292.33     176 2292.32
   196.7 2290.56   210.9 2291.16   230.2 2290.35     247 2290.56   251.5 2290.03
   255.6 2288.56   260.5 2288.04   267.9 2288.56     274 2289.34   278.5  2291.9
     283  2297.1   287.5 2301.47     292 2304.93     301  2313.2   308.5 2319.49
   315.4 2324.38   323.5 2328.53   374.8 2351.19   386.7 2357.05   422.4 2376.06
#Mann= 3 ,-1,0
       0      .1       0   255.6    .045       0   267.9      .1       0
#XS Ineff= 2 , 0
          212.99 2296.29
Permanent Ineff=
       F       F
Bank Sta=255.6,267.9
XS Rating Curve= 0 ,0
Exp/Cntr=0.3,0.1

Type RM Length L Ch R = 1 ,13500   ,284.2,283.7,281.7
XS GIS Cut Line= 4
2274504.56817908626065.0410501982274381.04018441626263.078093285
2274389.44244773626368.1176012682274466.99912871 626501.63256125
#Sta/Elev= 30
       0 2307.97    14.3 2304.71    49.7 2297.62    70.9 2293.83    81.7 2292.44
   122.3 2289.39   136.9 2288.94   194.9 2285.13   239.5 2284.45   253.1  2282.8
   275.6 2281.26   295.7 2281.36   303.7 2280.39   315.8 2280.87   323.7 2278.58
   327.4 2278.31     340 2280.32   353.3 2278.55   359.1 2276.62   367.3 2275.85
  371.13 2276.63   373.7 2278.32   382.5 2288.02   400.1  2302.5   411.4 2310.63
   429.3 2322.36   455.7  2335.8   467.4 2340.62   484.9 2348.82   493.2  2352.2
#Mann= 3 ,-1,0
       0      .1       0   359.1    .045       0  371.13      .1       0
Bank Sta=359.1,371.13
XS Rating Curve= 0 ,0
Exp/Cntr(USF)=0,0
Exp/Cntr=0.3,0.1

Type RM Length L Ch R = 1 ,13217   ,338.2,342.4,343
XS GIS Cut Line= 3
2274032.61853136626211.1498970222274135.74886003626410.897059935
   2274252.99176626611.729805255
#Sta/Elev= 30
       0 2301.87     7.8 2300.66    29.3 2293.94    47.3 2291.06    60.6  2286.1
    69.8 2280.49    90.2 2274.18   114.8  2271.1   155.3 2271.96   159.8 2271.14
   168.8 2267.56   190.9 2265.34     206 2269.19   213.9 2269.79   250.2 2268.64
  253.95 2267.63   267.7 2266.97   272.32267.627   278.4 2268.21   297.1 2267.47
   305.7 2268.22   343.2 2268.57   347.9 2269.69   355.5 2273.57   370.1 2283.78
   384.9 2295.96   399.3 2308.98     422 2326.42   434.4 2333.96   457.3 2345.21
#Mann= 3 ,-1,0
       0      .1       0  253.95    .045       0   272.3      .1       0
Bank Sta=253.95,272.3
XS Rating Curve= 0 ,0
Exp/Cntr(USF)=0,0
Exp/Cntr=0.3,0.1

Type RM Length L Ch R = 1 ,12874   ,250.4,251.4,249.6
XS GIS Cut Line= 3
2273845.98803659626392.2280539032273910.31884591626617.385886493
2273962.58762847 626841.20349389
#Sta/Elev= 30
       0 2279.41       8 2276.19    30.1 2265.31    34.3 2263.64    38.4 2262.95
      64 2263.53   117.5 2258.84   168.1 2259.16   188.2 2258.45   217.3 2256.21
   246.3 2256.55   258.6 2257.31   266.8 2254.65  271.94 2253.65   279.1 2252.99
   287.4  2253.1   288.8 2253.68   291.5 2254.84   295.7    2261   298.8 2264.39
   312.1 2277.32   324.3 2287.31   338.6  2298.1   358.7 2314.89   370.7 2323.64
   381.8 2330.66   402.4 2340.91   431.1 2356.71   438.7 2360.05     464 2373.13
#Mann= 3 ,-1,0
       0      .1       0  271.94    .045       0   288.8      .1       0
Bank Sta=271.94,288.8
XS Rating Curve= 0 ,0
Exp/Cntr(USF)=0,0
Exp/Cntr=0.3,0.1

Type RM Length L Ch R = 1 ,12623   ,206.1,218.7,215.2
XS GIS Cut Line= 2
2273609.14505814626504.5275268112273793.79830709626930.421310679
#Sta/Elev= 30
       0 2269.15    11.9 2264.99    26.9 2257.75    35.6 2254.48    45.4 2251.88
    57.4 2250.66   118.4 2251.31   140.2 2252.46     162 2251.49   179.5 2249.51
   196.9 2250.15   215.7 2249.36   224.8 2250.14   231.8  2249.8   244.9 2250.93
   253.6  2249.8   264.3 2249.62  274.72 2248.38   291.7 2247.75   299.2 2248.37
   301.5  2248.5   306.9 2251.01   310.3 2253.84   323.3 2266.51   353.9 2290.98
   379.9 2313.57     389 2320.07   398.2 2327.49   410.5 2335.23   464.2 2359.97
#Mann= 3 ,-1,0
       0      .1       0  274.72    .045       0   299.2      .1       0
#XS Ineff= 2 , 0
          241.94 2256.88
Permanent Ineff=
       T       F
Bank Sta=274.72,299.2
XS Rating Curve= 0 ,0
Exp/Cntr=0.3,0.1

Type RM Length L Ch R = 1 ,12404   ,167.7,163.3,159.1
XS GIS Cut Line= 3
2273503.67663216 626528.826256322273541.78057465626586.470682138
2273579.88451714626851.244231238
#Sta/Elev= 30
       0 2274.13    26.6 2265.42    35.3  2263.6    51.7  2256.5      58 2255.59
    66.2 2251.76    69.1 2250.96      84 2248.97    96.1  2248.2   120.3 2247.84
   124.4 2247.22   132.5 2245.18   136.5 2244.74   152.7 2244.75   156.7  2242.7
   164.8 2242.42   168.6 2241.49     189 2240.75   193.1 2241.47   197.1  2242.4
   213.3 2244.58   241.6 2244.48   253.6 2245.77   269.9 2245.64   281.9 2244.88
   302.2 2245.03   326.4  2243.9   330.5 2244.44   334.5 2247.38   336.6 2249.42
#Mann= 3 ,-1,0
       0      .1       0   168.6    .045       0   193.1      .1       0
Bank Sta=168.6,193.1
XS Rating Curve= 0 ,0
Exp/Cntr(USF)=0,0
Exp/Cntr=0.3,0.1

Type RM Length L Ch R = 1 ,12241   ,262.6,264.7,266.2
XS GIS Cut Line= 3
2273306.84981994626570.0496474062273336.63260203626623.658655165
 2273528.7315465626975.095483812
#Sta/Elev= 30
       0  2285.7     3.6 2284.98    41.5 2272.22    91.6 2259.82   122.3 2248.64
   126.9 2247.21     136 2245.69   140.6 2243.85   145.1 2241.11   149.7 2239.82
   194.7 2238.93   203.6 2237.05   208.9 2236.98   212.4 2236.22   218.1 2235.59
  227.97 2236.22   231.7 2238.84   236.3 2239.92   245.4  2240.2   259.1 2239.04
   286.4 2238.85   295.5 2239.66   324.4 2239.72   354.8 2240.65   377.6 2242.02
   382.2 2244.13   408.1 2264.44   414.1 2268.56   427.7 2276.07   461.8 2291.56
#Mann= 4 ,-1,0
       0      .1       0   212.4    .045       0  227.97      .1       0
  361.33     .06       0
Bank Sta=212.4,227.97
XS Rating Curve= 0 ,0
Exp/Cntr=0.3,0.1

Type RM Length L Ch R = 1 ,11976   ,161.8,159.2,160.9
XS GIS Cut Line= 3
2273165.62627058626619.6895037972273257.75017612626837.046654776
2273467.44093849627015.554784579
#Sta/Elev= 30
       0 2289.14    97.2 2265.75   114.6 2260.84   123.3 2255.03   128.2 2250.85
   137.3 2241.68   149.3 2231.94  158.42 2227.98   164.8 2227.01   170.5 2227.96
   184.1 2230.25   192.3 2229.37   201.3 2230.47   210.2 2229.92   227.5 2232.84
   236.3 2233.38   265.5 2233.09   328.8 2235.67   341.2 2234.98   354.8 2236.23
   378.2 2236.06   417.9 2237.41   428.4 2238.74   433.7 2240.27   439.4 2242.73
   459.9 2254.33   470.4 2261.23   483.1  2268.6   501.6 2277.76   511.5 2281.93
#Mann= 5 ,-1,0
       0      .1       0  158.42    .045       0   170.5      .1       0
  316.07     .06       0  466.07      .1       0
Bank Sta=158.42,170.5
XS Rating Curve= 0 ,0
Exp/Cntr(USF)=0,0
Exp/Cntr=0.3,0.1

Type RM Length L Ch R = 1 ,11817   ,170.3,169.1,166
XS GIS Cut Line= 3
2273006.04372085626671.3111065072273136.55839749626907.254305845
2273328.23991255627138.501206251
#Sta/Elev= 30
       0 2299.96    29.2 2291.42    61.6 2280.34    93.6 2267.57   116.4 2261.13
   126.6 2256.82   143.8 2252.83   148.4 2250.31   169.7 2232.92   185.4  2226.5
   189.6  2225.6     217 2223.27   230.7 2224.77  236.92 2223.24   241.3 2222.53
   250.32223.241   253.6 2224.11     259 2228.04   261.9 2228.57   313.7 2228.51
   333.2 2230.15     373 2230.87   435.5 2229.94   485.2 2233.35   490.3  2234.6
     498 2237.94   516.3 2248.36   526.4 2252.67   547.5 2265.02     570  2276.7
#Mann= 5 ,-1,0
       0      .1       0  236.92    .045       0   250.3      .1       0
  369.64     .06       0  499.64      .1       0
Bank Sta=236.92,250.3
XS Rating Curve= 0 ,0
Exp/Cntr(USF)=0,0
Exp/Cntr=0.3,0.1

Type RM Length L Ch R = 1 ,11648   ,123.7,124.7,126.4
XS GIS Cut Line= 4
2272863.72580315626769.1742012592272946.83057853626879.672728639
2273006.17275979626929.8210508312273277.92126502627145.568043169
#Sta/Elev= 30
       0 2288.53    20.3  2282.2    60.3 2267.05    70.1 2266.03    80.1 2260.59
    93.9 2258.72   105.1 2254.89   113.9 2253.08   120.5  2250.1   133.8    2248
   140.3 2243.55   165.8 2220.27   171.4 2216.74  173.98 2216.23   181.9 2215.75
   185.7 2216.24   194.2  2221.1   208.8  2223.9   223.6  2225.1   227.8 2225.07
   234.2 2223.05     244 2224.77   285.7 2226.15   330.9 2226.03   388.6 2227.49
   433.3 2226.58   461.8 2227.67   504.5 2231.59   518.7 2237.53   562.9 2261.98
#Mann= 5 ,-1,0
       0      .1       0  173.98    .045       0   185.7      .1       0
  435.96     .06       0  562.93      .1       0
Bank Sta=173.98,185.7
XS Rating Curve= 0 ,0
Exp/Cntr(USF)=0,0
Exp/Cntr=0.3,0.1

Type RM Length L Ch R = 1 ,11523   ,146.5,147,147.7
XS GIS Cut Line= 4
2272746.93351667626817.246738742     2272893.816      626997.638
2273007.84437054627142.1156147772273196.48360558627232.493165963
#Sta/Elev= 30
       0 2287.26   108.9 2261.26   139.2 2253.44   148.7 2248.28   166.7 2242.61
     173 2239.39   180.5 2233.87   191.3  2223.7     197 2219.58   201.1 2218.39
   216.9 2218.45   221.7 2216.85     2272213.662   236.4 2212.78   241.42213.646
   242.9  2214.4   248.2 2219.38   253.9 2221.19   277.9 2220.13   362.1 2221.41
   393.5 2220.76   474.7 2226.95   503.2 2229.88   524.2 2231.07   542.2 2233.33
   554.2 2233.02   572.2 2234.92   578.2 2236.61   598.9 2245.25   625.9 2258.28
#Mann= 5 ,-1,0
       0      .1       0     227    .045       0   241.4      .1       0
  506.68     .06       0  606.68      .1       0
Bank Sta=227,241.4
XS Rating Curve= 0 ,0
Exp/Cntr=0.3,0.1

Type RM Length L Ch R = 1 ,11376   ,191.7,190.6,188.3
XS GIS Cut Line= 3
2272677.28233037626933.5862845472272870.77228988627229.875178613
2273034.48750838627284.258339262
#Sta/Elev= 30
       0 2274.52    13.4 2270.56    80.7 2252.38   100.4 2247.77   107.7 2246.42
   118.9  2245.1   123.7 2244.25   126.1 2243.37     129 2241.91   133.3 2238.33
   142.8 2228.36   152.4 2217.64   157.2 2212.78   161.62210.767   166.7 2209.94
   171.5 2209.83   181.22210.593   185.8 2212.78   190.6 2216.97   195.4 2218.34
   201.2 2217.56   224.1 2216.56   247.5 2216.42   271.8 2215.34   305.3 2215.38
   319.7 2216.19   353.9 2216.65   436.7 2220.57   464.5 2223.04   526.4 2229.53
#Mann= 4 ,-1,0
       0      .1       0   161.6    .045       0   181.2      .1       0
  503.87     .06       0
Bank Sta=161.6,181.2
XS Rating Curve= 0 ,0
Exp/Cntr(USF)=0,0
Exp/Cntr=0.3,0.1

Type RM Length L Ch R = 1 ,11185   ,132.3,130,125.2
XS GIS Cut Line= 3
2272503.58914523627047.5724372962272664.32836352627238.233232312
2272999.63379726627344.608937034
#Sta/Elev= 30
       0  2273.8   117.2  2247.1   127.7 2244.16   132.1 2242.55     135  2240.8
   148.6 2229.22   157.7 2222.66   169.5 2215.22   174.8 2213.81   194.6 2212.83
   199.5 2210.09   205.9 2204.62  207.88 2204.08   211.9 2203.31   220.1 2203.43
     223 2204.06   225.8 2205.97   231.5 2211.41   234.3 2212.52   236.7 2212.78
   257.6 2212.66   295.4 2210.74   316.4 2211.87   337.6 2211.81   369.5 2213.79
   412.9 2214.84   433.9 2216.22   493.7 2217.37   531.9 2219.76   601.2 2226.63
#Mann= 4 ,-1,0
       0      .1       0  207.88    .045       0     223      .1       0
  589.38     .06       0
Bank Sta=207.88,223
XS Rating Curve= 0 ,0
Exp/Cntr=0.3,0.1

Type RM Length L Ch R = 1 ,11055   ,163.8,160.6,156.7
XS GIS Cut Line= 4
2272405.64548805 627214.028406392272523.85335016627298.462593611
2272596.62812856627326.8286015182272878.81164406627464.986082863
#Sta/Elev= 30
       0 2245.16    57.2 2237.57    67.2 2232.84    81.1 2223.41   101.8 2213.04
   107.3 2211.44   140.7 2207.31     180 2207.82   184.2 2207.17   188.5 2205.47
   192.8 2201.74  195.62 2200.41   201.4 2199.73   207.8 2200.38   218.8 2205.56
   227.3 2206.97   249.6 2205.35   290.6 2205.67     303 2206.64   338.7 2205.85
   360.9 2207.45     383 2210.11   396.6 2210.72   437.9 2212.02   474.3 2211.75
   490.1 2214.16   510.7 2218.95   521.3 2223.39   530.2 2224.53   537.6 2227.04
#Mann= 7 ,-1,0
       0      .1       0     110     .05       0  195.62    .045       0
   207.8     .05       0  215.27      .1       0  333.37     .06       0
  433.37      .1       0
Bank Sta=195.62,207.8
XS Rating Curve= 0 ,0
Exp/Cntr(USF)=0,0
Exp/Cntr=0.3,0.1

Type RM Length L Ch R = 1 ,10895   ,203,208.4,212.5
XS GIS Cut Line= 4
  2272367.497556627322.9548259392272519.75780724 627478.25098458
2272575.73299431627468.9155143952272804.81465492627557.959808801
#Sta/Elev= 30
       0 2228.65    14.3 2227.01    18.1 2225.95    23.8 2222.86    31.1 2217.25
    38.8 2213.19    55.8 2206.78    69.5 2203.76   166.7 2202.06   211.4  2201.8
     226 2202.34   230.1 2202.15   232.7 2201.17     241 2196.39   246.6  2195.7
  254.74 2196.39   260.5 2199.19   270.6  2202.8   274.8 2203.58   291.9  2201.8
   300.5 2202.39   313.3 2204.53   361.3 2204.28   404.6 2206.33   426.2  2206.6
   437.8 2207.58   463.3 2212.73   494.2 2222.46   502.2 2223.77     520 2229.18
#Mann= 6 ,-1,0
       0      .1       0     180     .06       0     241    .045       0
  254.74     .06       0  294.23     .07       0  394.23     .06       0
Bank Sta=241,254.74
XS Rating Curve= 0 ,0
Exp/Cntr(USF)=0,0
Exp/Cntr=0.3,0.1

Type RM Length L Ch R = 1 ,10686   ,221,220,218.7
XS GIS Cut Line= 4
2272251.21662754627456.157299599 2272406.9003096627606.823400423
2272449.52638346627633.5691722582272631.45223009627702.673897224
#Sta/Elev= 30
       0 2218.67      13 2217.49    24.5 2214.99    29.2 2212.59    43.8 2202.93
    47.5 2201.17    52.3 2199.79    64.7 2198.78    76.2 2199.08    86.3 2198.19
     170 2197.75     185 2197.41   193.8  2196.4   222.2  2196.2   227.6 2194.48
   236.1 2190.38   243.7 2189.81  251.59 2190.41   260.7 2194.24   277.1 2197.58
   310.9 2196.18   325.4 2196.78   355.4 2199.24   367.3  2198.8   381.1 2199.78
   392.8 2199.78   436.2 2205.41   453.8 2209.57   458.1 2209.39   461.6  2210.4
#Mann= 8 ,-1,0
       0      .1       0      30     .06       0      60      .1       0
     170     .06       0     200     .05       0   236.1    .045       0
  251.59     .05       0  316.97     .06       0
Bank Sta=236.1,251.59
XS Rating Curve= 0 ,0
Exp/Cntr=0.3,0.1

Type RM Length L Ch R = 1 ,10466   ,82,86,89
XS GIS Cut Line= 4
2272174.96338357627544.0892077952272350.06554445627819.117964369
2272403.29416119627847.5393316292272642.86933339627886.545190272
#Sta/Elev= 30
       0 2214.38    39.2 2209.09    62.9 2202.47    76.7 2197.14    84.2 2195.83
     132 2193.25   186.2  2193.1   317.5 2190.11   328.4 2190.65     335 2189.13
  342.72 2185.17   346.9 2183.96   352.8 2185.15   361.6 2188.89   364.7 2189.15
   378.3  2187.5   387.3 2190.76   395.4 2191.66   403.5 2191.58   411.6 2190.31
   433.9 2189.73   468.3 2191.47     492 2193.82   504.8 2196.98   525.1  2203.4
   538.4 2205.89   553.4 2209.98   569.6 2211.74   577.7  2216.1   629.1 2231.04
#Mann= 8 ,-1,0
       0      .1       0      40     .06       0  342.72    .045       0
   352.8     .06       0  376.04     .07       0  476.38     .06       0
  516.38     .07       0  576.38      .1       0
#XS Ineff= 2 , 0
                          366.03         2194.32
Permanent Ineff=
       F       F
Bank Sta=342.72,352.8
XS Rating Curve= 0 ,0
Exp/Cntr(USF)=0,0
Exp/Cntr=0.3,0.1

Type RM Length L Ch R = 1 ,10380   ,51.6,51,51.7
XS GIS Cut Line= 5
2272112.01540907 627743.943967062272313.29010818627860.072427492
2272360.71724379627951.3854716342272360.09520889627991.293870561
2272563.09040554628058.273018621
#Sta/Elev= 30
       0 2198.54     9.4 2196.77    27.9 2196.17    37.1 2194.84    50.8 2191.41
    64.8 2190.11     165 2189.86   188.4 2189.24   200.2 2187.54   212.6 2187.12
   232.4 2187.93   238.6 2187.18   270.9 2186.33   274.2 2185.72   281.52182.736
   288.7 2182.18   293.9 2182.76   310.2 2186.27   375.2 2185.15   414.7 2185.65
     430 2186.72   442.7 2190.57   476.4 2196.23   493.2  2198.8   503.4 2198.65
   514.3 2203.92   525.6  2204.1   531.1 2205.11   563.6 2218.14   588.9 2230.44
#Mann= 7 ,-1,0
       0     .06       0      50     .07       0     210     .06       0
  242.37     .07       0   281.5    .045       0   293.9     .07       0
  515.18      .1       0
#XS Ineff= 2 , 0
                           332.2         2190.39
Permanent Ineff=
       F       F
Bank Sta=281.5,293.9
XS Rating Curve= 0 ,0
Exp/Cntr(USF)=0,0
Exp/Cntr=0.3,0.1

Type RM Length L Ch R = 1 ,10329   ,134.7,136.5,138.3
XS GIS Cut Line= 5
2272076.05133476627769.7723313012272277.32603387627885.900791733
2272324.75316948627977.2138358752272324.13113458628017.122234802
2272527.12633123628084.101382862
#Sta/Elev= 30
       0 2199.49    46.3 2197.29      74 2192.13   101.7  2189.6   120.2 2188.91
   206.9 2188.61   226.4 2187.48   289.7 2185.63   294.7  2184.7   302.2 2181.68
     308 2180.79  314.78 2181.68   322.9 2185.04   328.9 2185.65   375.2  2184.5
   404.7 2184.98   417.3 2184.28   472.1 2185.38   476.3 2186.58   484.7  2193.3
     489 2194.76   498.8 2196.83     510 2195.86   514.2  2197.4   522.7 2202.66
   526.9 2204.12   539.5 2203.49   546.3 2204.47   574.8 2215.05   588.9 2221.29
#Mann= 6 ,-1,0
       0     .06       0      30     .07       0   302.2    .045       0
  314.78     .07       0  525.18     .06       0  555.18      .1       0
Bank Sta=302.2,314.78
XS Rating Curve= 0 ,0
Exp/Cntr(USF)=0,0
Exp/Cntr=0.3,0.1

Type RM Length L Ch R = 1 ,10193   ,174.4,170.6,160.7
XS GIS Cut Line= 4
2272043.88742642627783.2699102532272244.40956698628036.539306438
2272258.96275913628088.2472934652272449.34534107628198.606785126
#Sta/Elev= 30
       0 2198.52    39.1 2196.68    48.4 2195.33      79 2194.64    84.2 2193.78
    99.4 2187.34     110 2186.24     168  2186.6   186.1 2186.17   206.5 2184.78
   226.9 2184.61   266.4 2183.13   306.2 2182.58     332 2183.29   352.22177.772
   356.9 2177.22   365.3 2177.76   373.6 2182.14   396.7 2181.07   413.4 2181.06
   456.8 2181.62   463.2 2182.44   470.6  2181.4   475.3 2183.88   484.5 2190.96
   489.5 2193.58   526.1 2201.14   544.6  2203.6   562.7 2209.68   596.8 2218.74
#Mann= 8 ,-1,0
       0     .06       0      90     .07       0     110     .06       0
   352.2    .045       0   365.3      .1       0  416.76     .08       0
  526.76     .06       0  536.76      .1       0
Bank Sta=352.2,365.3
XS Rating Curve= 0 ,0
Exp/Cntr(USF)=0,0
Exp/Cntr=0.3,0.1

Type RM Length L Ch R = 1 ,10022   ,151.9,149.9,144.5
XS GIS Cut Line= 4
2271920.80400928627876.7823418222272065.05591333628079.053434397
2272146.36228547628105.3932710092272340.13534509628220.105283738
#Sta/Elev= 30
       0 2196.26    44.7 2192.31    62.9 2185.22    74.2 2183.26    85.9  2183.3
   114.5 2181.63   128.9 2182.42     143  2181.3   162.6 2182.54   191.8  2181.9
     197 2182.62   211.7 2182.02   216.7 2182.51   233.1 2180.33     259 2179.68
   268.5 2177.29  275.98 2172.93   281.1 2172.16   289.6 2172.94   320.2 2177.73
   363.9 2179.32   387.1 2178.94   410.4 2177.23   489.4 2178.74   494.1 2178.61
   498.7 2177.38   517.3 2178.22   530.7 2184.61   549.8 2196.91   559.1 2201.75
#Mann= 6 ,-1,0
       0     .06       0     110     .05       0     140     .06       0
  275.98    .045       0   289.6      .1       0  453.91     .06       0
Bank Sta=275.98,289.6
XS Rating Curve= 0 ,0
Exp/Cntr(USF)=0,0
Exp/Cntr=0.3,0.1

Type RM Length L Ch R = 1 ,9872    ,145.2,150.9,156.4
XS GIS Cut Line= 4
2271852.69170917628091.0399253272272104.33876571628234.513233192
2272175.07124118628218.7585311042272327.21933977 628293.05060027
#Sta/Elev= 30
       0 2183.58    22.4 2178.39    36.2 2175.92    40.8 2175.61    54.7 2175.51
   100.9 2177.26   137.5 2176.72   191.8 2177.08   206.2 2176.32   235.8 2173.47
   297.4 2172.48   300.7 2171.57   305.9 2169.19   309.82168.458   318.2 2167.67
   322.3 2167.74  323.46 2168.48   326.4 2170.37   330.5 2174.85   334.2  2176.1
   363.4 2178.34   413.2 2175.04   447.9 2174.26   465.7 2175.31   469.5 2177.81
   475.4 2186.04   479.1 2189.22   511.3 2209.35   523.6 2216.52   531.5 2220.57
#Mann= 7 ,-1,0
       0     .06       0      60     .05       0     280      .1       0
   309.8    .045       0  323.46      .1       0  392.14     .06       0
  502.14      .1       0
Bank Sta=309.8,323.46
XS Rating Curve= 0 ,0
Exp/Cntr(USF)=0,0
Exp/Cntr=0.3,0.1

Type RM Length L Ch R = 1 ,9721    ,191.7,187.9,184.8
XS GIS Cut Line= 2
2271837.98202968628129.8404208732272218.45095553628456.381332202
#Sta/Elev= 30
       0 2178.89    17.4 2175.85    29.2 2175.19      82 2175.34   150.5 2174.71
   162.8 2175.11   189.4 2174.48   196.8 2175.36   207.8 2173.98   261.2  2172.2
   304.6  2168.4     316 2168.64   327.3 2169.61   341.5 2169.65   355.2 2165.94
   365.62165.422   372.7 2164.98   377.1 2165.44   379.8  2166.9     384 2170.32
   386.9 2171.69   408.8 2171.45   412.4 2172.11   415.2 2174.43   419.3 2180.61
   423.7 2185.68   429.4 2190.61   445.7  2201.7   461.5 2210.37   501.4 2229.92
#Mann= 6 ,-1,0
       0     .06       0      60     .05       0     340     .06       0
   365.6    .045       0   377.1     .06       0     470      .1       0
Bank Sta=365.6,377.1
XS Rating Curve= 0 ,0
Exp/Cntr(USF)=0,0
Exp/Cntr=0.3,0.1

Type RM Length L Ch R = 1 ,9535    ,187,192.7,197.1
XS GIS Cut Line= 4
2271668.12454869628311.9207932522271965.59507431628481.911622672
2272039.14594686 628494.448703222272178.15782972628535.944992652
#Sta/Elev= 30
       0 2177.36    23.1 2175.22    46.1 2169.62    69.2 2168.01   115.2 2168.41
   198.2 2165.76   239.6 2167.37   279.5 2165.92   294.1 2166.93     300 2166.46
   341.1 2165.97   361.5 2166.54   365.5 2164.68   369.6 2161.81   373.6  2161.3
   381.8 2160.92  386.52 2161.29   393.9 2164.22     402  2164.7   410.1 2167.02
   418.3 2168.23     446 2169.36   464.2 2171.68   468.3 2174.26   472.6 2178.97
   476.7 2182.57   481.3 2185.62   501.8  2195.5   535.2 2212.77   562.3 2225.26
#Mann= 8 ,-1,0
       0     .06       0      40     .05       0     100     .06       0
     270     .05       0     300     .06       0   373.6    .045       0
  386.52     .06       0  477.23      .1       0
Bank Sta=373.6,386.52
XS Rating Curve= 0 ,0
Exp/Cntr=0.3,0.1

Type RM Length L Ch R = 1 ,9345    ,256.7,253.1,248.7
XS GIS Cut Line= 4
2271595.18336556628436.6502390692271875.02238606628583.806965369
2271907.89041297628650.7436475052272027.85759707628711.192173166
#Sta/Elev= 30
       0 2169.71    23.7 2165.06    41.8 2163.76    95.7 2164.68   112.9 2164.51
   119.6 2163.85   146.3 2164.43   186.4 2162.12   213.5 2161.49     241 2159.08
   267.7 2159.15   317.7 2161.07   348.9 2159.85   353.4 2159.08   357.8 2157.07
  370.78 2156.02   375.6 2155.31   380.1 2156.02   384.5 2157.87   404.5  2160.1
   431.5 2160.17   435.9 2161.29   440.3 2163.67   455.3 2169.85   467.2 2172.85
   476.2 2174.06   485.2 2174.42     503 2177.64   516.5 2178.63   525.1 2178.54
#Mann= 6 ,-1,0
       0     .05       0      50     .06       0     260     .05       0
  370.78    .045       0   380.1     .06       0  490.74      .1       0
Bank Sta=370.78,380.1
XS Rating Curve= 0 ,0
Exp/Cntr(USF)=0,0
Exp/Cntr=0.3,0.1

Type RM Length L Ch R = 1 ,9092    ,139.6,139.5,138.8
XS GIS Cut Line= 2
2271403.50692968628578.6153955522271935.24727973628857.572352466
#Sta/Elev= 30
       0 2168.72    57.2 2163.57    74.4 2161.41    91.6 2158.13   100.1 2157.28
   145.3 2156.45     195 2157.31   231.1 2156.37   255.2 2156.72   304.6 2155.95
   307.9 2155.56   316.9 2149.45   322.4  2148.8   329.3 2149.44     335 2150.66
   339.5 2150.81   353.1 2150.06   362.1 2150.34   375.7 2151.69   389.2 2154.28
   411.3  2153.5   426.1 2154.78   443.8 2154.14     475 2154.83   514.9 2157.65
   535.7 2157.97   542.8 2159.27     548  2159.5   556.6    2162   600.5 2187.01
#Mann= 8 ,-1,0
       0     .05       0     120     .06       0   316.9    .045       0
   329.3     .06       0     340      .1       0     380     .05       0
     450     .06       0     560      .1       0
Bank Sta=316.9,329.3
XS Rating Curve= 0 ,0
Exp/Cntr(USF)=0,0
Exp/Cntr=0.3,0.1

Type RM Length L Ch R = 1 ,8953    ,234,234.6,236.8
XS GIS Cut Line= 3
2271266.78885807628692.316748641 2271717.9949196 628885.23431064
2271874.39360754628966.721150159
#Sta/Elev= 30
       0 2166.26    97.2 2159.95     132 2156.38     153 2154.85   188.6 2153.45
   239.4 2152.95   248.5 2152.43   321.7 2152.36   340.8 2152.77   362.6 2151.68
   388.8 2151.47   413.1 2149.93   426.82146.253   434.4 2145.28   439.7 2146.23
   445.2 2148.81   449.6 2149.97   462.6 2151.04   510.1 2151.41   524.9 2152.25
   557.5 2151.21   585.8 2151.79   605.9 2153.22   628.5 2153.61     633 2155.61
   640.6 2161.41   646.4 2164.76   655.5 2171.77   664.3 2177.33   667.1 2179.67
#Mann= 7 ,-1,0
       0     .08       0      50     .05       0     160     .06       0
     410     .05       0   426.8    .045       0   439.7     .05       0
  590.72     .06       0
Bank Sta=426.8,439.7
XS Rating Curve= 0 ,0
Exp/Cntr(USF)=0,0
Exp/Cntr=0.3,0.1

Type RM Length L Ch R = 1 ,8719    ,207.4,208.3,209.2
XS GIS Cut Line= 4
2271233.32263303628755.2526319842271573.30475188629055.094775409
2271625.17148684629097.6799513642271761.79650414629142.032290159
#Sta/Elev= 30
       0 2164.34    85.6  2159.3   105.4 2157.49   137.1 2152.92   169.1 2150.55
   215.9  2149.5   227.3 2148.68   307.8 2147.61   361.1 2145.34     402 2146.98
   451.8 2145.06   475.5 2145.58   477.7 2145.16   482.9 2142.43   493.3 2140.82
   498.4 2139.82  504.64 2140.82   510.8 2144.43   516.5 2146.03     553 2145.32
   585.9 2147.99   599.3 2147.53   616.1 2149.53   624.5 2153.45   627.2 2155.75
   630.4 2159.51   637.1 2170.05   641.3 2174.72   652.6  2184.3   664.1  2191.5
#Mann= 5 ,-1,0
       0     .05       0     150     .06       0     300     .05       0
   493.3    .045       0  504.64     .06       0
Bank Sta=493.3,504.64
XS Rating Curve= 0 ,0
Exp/Cntr(USF)=0,0
Exp/Cntr=0.3,0.1

Type RM Length L Ch R = 1 ,8510    ,144.3,145.4,145.7
XS GIS Cut Line= 3
2271232.41806004628820.5495958592271414.39854576629174.790359242
2271592.78466213629354.094078609
#Sta/Elev= 30
       0 2160.63    45.7  2157.2    86.4 2150.55   110.2 2148.61   181.5 2146.38
   225.6 2146.36     257 2143.95   297.5 2143.81   324.5 2142.23   351.5 2139.19
   384.6 2140.71   412.9 2140.17   457.5 2141.22   474.7 2140.72   480.4 2139.93
   488.9 2135.79   508.8 2135.65   514.5 2134.41   523.12135.635     537 2139.52
   568.1 2139.84   582.2 2143.78   593.5 2143.88   604.9 2142.84   610.4 2144.83
   616.2 2148.35   627.3 2157.12   638.6  2164.4   644.2 2166.93   651.2 2168.45
#Mann= 7 ,-1,0
       0     .05       0     170     .06       0     260     .05       0
   508.8    .045       0   523.1     .05       0  528.25     .07       0
  638.25     .06       0
Bank Sta=508.8,523.1
XS Rating Curve= 0 ,0
Exp/Cntr=0.3,0.1

Type RM Length L Ch R = 1 ,8365    ,153.7,154.3,153.4
XS GIS Cut Line= 2
2271065.76514127628962.2620981682271451.67101123629423.278245416
#Sta/Elev= 30
       0 2153.34       9 2153.24    29.3 2151.65      56 2149.35   100.1 2144.51
   134.6 2142.24   181.2 2140.97     249 2140.15   285.5 2138.18   324.2 2137.98
   346.5 2137.06     390 2136.59   433.7 2134.52   447.2 2136.01   460.9 2136.68
   464.9 2135.97  471.04 2132.18   473.3 2131.19   477.4 2130.91   484.32132.167
   492.2 2132.81   504.6 2136.51   509.8 2137.32   556.7 2135.62   568.8 2135.89
   574.5 2137.39     583 2141.75   589.5 2144.29   594.4 2145.72   601.2 2146.69
#Mann= 7 ,-1,0
       0     .06       0      80     .05       0     230     .06       0
     370     .05       0  471.04    .045       0   484.3     .05       0
     500     .06       0
Bank Sta=471.04,484.3
XS Rating Curve= 0 ,0
Exp/Cntr(USF)=0,0
Exp/Cntr=0.3,0.1

Type RM Length L Ch R = 1 ,8210    ,113.8,113.1,112.1
XS GIS Cut Line= 3
2271078.32165875629032.225600455 2271238.2107413629404.210081355
2271335.84877669 629515.41406891
#Sta/Elev= 30
       0 2148.12    14.1 2146.65    48.9 2141.14    78.3 2139.33    96.8 2138.79
   145.3 2139.52   166.8 2138.76   176.9 2137.51   190.9 2137.36   203.1 2136.51
   231.8 2135.85     271 2135.98   288.3 2135.16   331.9 2134.43   376.7  2132.8
   432.5  2131.3   443.4 2128.74   452.3 2128.27  457.98 2128.73   463.7 2129.48
   470.1 2129.74   475.4    2131   480.6 2131.72     502 2131.72   523.3  2133.3
   528.6 2135.61   535.2  2139.8   541.2 2144.21   549.9 2149.59   552.9 2151.01
#Mann= 7 ,-1,0
       0     .06       0      20     .05       0     130     .06       0
   443.4    .045       0  457.98     .06       0  464.89     .05       0
  514.89     .06       0
Bank Sta=443.4,457.98
XS Rating Curve= 0 ,0
Exp/Cntr(USF)=0,0
Exp/Cntr=0.3,0.1

Type RM Length L Ch R = 1 ,8097    ,122.8,121.2,119.9
XS GIS Cut Line= 3
2270965.17477068629319.6956269582271192.80728193629521.159349312
2271257.70122707629574.182450824
#Sta/Elev= 30
       0 2135.12      40 2133.19      57 2131.89    62.8 2131.12    78.8 2131.93
    89.5 2131.37    99.5 2131.35   121.5  2130.5   164.3 2131.02   181.7  2129.9
   196.3 2129.81   217.7 2128.63   249.7 2127.66   263.9 2128.64   272.4 2129.83
   279.9  2129.9   281.8 2129.38   286.8 2126.31   292.2 2125.68  299.94 2126.29
   306.4 2127.49   312.1    2129     323 2130.29     329 2131.94   334.2 2134.57
     349 2143.19   367.2 2153.18   374.6 2155.94   379.9 2157.47   387.8 2157.86
#Mann= 5 ,-1,0
       0     .06       0     190     .05       0   286.8    .045       0
  299.94     .05       0  343.98      .1       0
#XS Ineff= 2 , 0
          274.96 2132.69
Permanent Ineff=
       T       F
Bank Sta=286.8,299.94
XS Rating Curve= 0 ,0
Exp/Cntr=0.3,0.1

Type RM Length L Ch R = 1 ,7976    ,106.7,103.4,99.3
XS GIS Cut Line= 3
2270869.31802524629354.4449432182271077.06513422629585.638658748
2271181.40441515629637.995589722
#Sta/Elev= 30
       0 2139.44    52.2 2135.75    80.4 2132.57   111.6 2129.87   137.1 2129.02
     165 2127.44   177.8 2127.74   201.8 2126.02   237.7 2125.36     251 2125.77
   267.2    2127   301.4 2126.44   314.3 2128.42   321.7 2128.69   324.7 2127.85
   330.7 2123.83   332.2 2122.87   336.6 2122.13   342.6  2123.7   350.1 2125.48
   354.6 2129.71   359.1 2136.21   360.5 2137.71     377 2153.41   385.9    2160
   394.9  2164.6   399.3 2166.24   408.3 2167.31   417.1 2166.56   427.6 2163.56
#Mann= 7 ,-1,0
       0     .05       0      70     .06       0     220     .05       0
     260     .07       0   330.7    .045       0   342.6     .07       0
  350.82     .05       0
#XS Ineff= 2 , 0
           267.1 2131.62
Permanent Ineff=
       T       F
Bank Sta=330.7,342.6
XS Rating Curve= 0 ,0
Exp/Cntr(USF)=0,0
Exp/Cntr=0.3,0.1

Type RM Length L Ch R = 1 ,7873    ,60.6,55.7,53.3
XS GIS Cut Line= 3
2270865.77666565629509.9686078222271026.06244432629714.444788497
2271152.09369016629684.675633229
#Sta/Elev= 30
       0 2130.55     6.8 2130.29    18.2 2129.27    38.2 2126.84      61 2125.74
    81.7 2125.54   100.6  2125.8   143.6  2124.8   159.5 2125.09   250.3 2124.95
   269.3 2124.77   278.4 2124.18   290.8 2125.62   303.1 2126.29   307.2 2125.99
   315.4 2122.48   322.5 2120.33   327.7  2119.9   331.9 2120.31     336 2122.11
   340.1  2124.9   344.2 2126.74   348.3 2130.75   352.4 2135.96   356.5 2139.28
   368.8 2147.25   377.1  2151.2   381.2 2152.51   385.3 2153.29   389.3 2153.13
#Mann= 6 ,-1,0
       0     .05       0      80     .06       0     240     .07       0
   322.5    .045       0   331.9     .07       0  349.81     .06       0
Bank Sta=322.5,331.9
XS Rating Curve= 0 ,0
Exp/Cntr(USF)=0,0
Exp/Cntr=0.3,0.1

Type RM Length L Ch R = 1 ,7817    ,49.8,50.2,49.6
XS GIS Cut Line= 3
2270690.19914296629588.5846979082271072.13606827629783.502809301
2271170.48125622629690.621242908
#Sta/Elev= 30
       0 2131.85    25.7 2129.79    69.6 2127.42    96.5  2123.5   105.5 2122.95
     128 2122.57   204.1 2123.37   213.3 2123.01   231.2 2120.85   238.9 2120.42
   257.6  2120.7   276.2 2122.41   293.3 2123.06     330 2122.92     370  2123.3
   397.3 2123.21   433.3 2125.41   455.9 2125.36   458.8 2124.07   464.4  2120.2
   467.1 2118.69   470.1 2118.52     473 2118.64   478.4 2120.23   487.1 2124.64
   494.9 2130.11   500.4 2132.49   522.4  2139.3   538.9  2141.7   564.1 2143.64
#Mann= 9 ,-1,0
       0     .06       0      40     .05       0     120     .06       0
     150     .05       0     260     .06       0     330     .07       0
     370     .06       0   464.4    .045       0   478.4     .06       0
#XS Ineff= 2 , 0
           313.4 2129.02
Permanent Ineff=
       F       F
Bank Sta=464.4,478.4
XS Rating Curve= 0 ,0
Exp/Cntr(USF)=0,0
Exp/Cntr=0.3,0.1

Type RM Length L Ch R = 1 ,7767    ,37.5,39.3,56.4
XS GIS Cut Line= 3
 2270672.0042794629647.4375695052271101.44094751629826.715088853
2271207.23652848629715.952579197
#Sta/Elev= 30
       0 2129.66    13.2 2128.58    43.5  2127.9    69.5 2126.16   105.4 2121.56
   121.6 2121.16   194.1 2121.99   216.9 2119.63     240  2119.8   264.4 2121.15
   288.9 2120.73     360 2123.02   409.5 2122.25   433.6 2124.69   442.3 2124.99
     451 2124.44   459.6 2120.63     464 2119.98   482.5 2121.06   496.7 2121.15
   499.5  2120.5   505.12117.646   510.8 2116.43   515.62117.671   517.3 2118.53
   522.1 2122.36   530.6 2125.74   556.2 2128.86   590.9 2134.14   618.5 2137.46
#Mann= 7 ,-1,0
       0     .06       0     160     .05       0     240     .06       0
     270     .07       0     370     .06       0   505.1    .045       0
   515.6     .06       0
#XS Ineff= 2 , 0
          269.87 2125.33
Permanent Ineff=
       T       F
Bank Sta=505.1,515.6
XS Rating Curve= 0 ,0
Exp/Cntr(USF)=0,0
Exp/Cntr=0.3,0.1

Type RM Length L Ch R = 1 ,7727    ,109.8,111.1,105.8
XS GIS Cut Line= 4
2270665.24485025629662.5399973032271096.97312631629842.188983838
2271207.93593954 629809.470036022271241.39484363629744.326838094
#Sta/Elev= 30
       0 2129.18    29.2 2127.99   107.2 2121.03   124.5 2120.74   193.8 2121.42
   209.2  2119.5   215.1 2119.25   245.8 2119.63   263.1  2120.6   285.7 2120.27
   310.8 2121.56   349.8 2122.47   410.4 2121.77   427.8 2123.84   440.8 2124.02
   445.1 2123.79     454 2120.99   462.4 2119.41   493.5  2119.2   527.8 2116.05
     546 2115.47  560.54 2116.05   583.3 2116.47   588.1 2116.16   592.6 2116.74
   604.5  2122.5   613.4 2124.93   633.1 2133.07   642.1 2136.08   656.5 2141.91
#Mann= 9 ,-1,0
       0     .06       0     170     .05       0     200     .06       0
     270     .07       0     380     .06       0     460     .07       0
  487.61     .06       0   527.8    .045       0  560.54     .06       0
Bank Sta=527.8,560.54
XS Rating Curve= 0 ,0
Exp/Cntr(USF)=0,0
Exp/Cntr=0.3,0.1

Type RM Length L Ch R = 1 ,7615    ,109.2,118,124.7
XS GIS Cut Line= 4
2270658.31989618629674.3911345122271194.86106374629923.328300795
2271241.93469731629907.7687018042271343.86173873630003.125393873
#Sta/Elev= 30
       0 2128.97    54.7 2126.25    93.9 2122.02   116.7 2120.82   187.2 2120.66
   206.2 2119.23   235.8 2119.16   275.4 2120.48   292.7 2119.98   325.8 2121.37
   407.7 2120.92   429.8 2122.51   438.6 2122.22     465 2117.92   473.9 2118.23
   482.7 2119.62   567.4 2117.25   588.5 2118.85   601.3 2117.18   608.82114.355
   616.4 2113.18   622.4 2113.47   623.62114.283   630.8 2120.13   641.1 2122.64
   684.1 2121.52   698.9 2123.64   707.5 2127.33     737 2146.13   780.6 2170.04
#Mann= 9 ,-1,0
       0     .06       0     290     .07       0     390     .06       0
     400     .07       0     500     .06       0   608.8    .045       0
   623.6     .06       0  681.06      .1       0  741.06     .06       0
Bank Sta=608.8,623.6
XS Rating Curve= 0 ,0
Exp/Cntr(USF)=0,0
Exp/Cntr=0.3,0.1

Type RM Length L Ch R = 1 ,7494    ,106.5,106.2,104
XS GIS Cut Line= 3
2270657.94479012629679.3956621462271049.76699972 629869.91468385
2271242.44893683630083.905104061
#Sta/Elev= 30
       0 2128.93      15 2127.63    50.9 2126.23   104.8 2120.81   184.8 2120.22
   202.6 2119.18   233.8 2119.02   260.2 2119.75   287.3 2119.45   315.1 2121.08
   402.8 2120.49   424.9 2121.94     434 2121.65   445.5 2119.46   457.2 2119.09
   463.2 2117.43     468 2117.04   475.2 2117.32     485 2118.96   547.3 2116.59
     604 2117.17   609.6 2115.82   618.1 2110.06   623.8 2109.32  628.78 2110.06
   633.9 2113.07   642.5 2121.86   648.5 2125.91   683.3  2145.4   723.6 2169.14
#Mann= 9 ,-1,0
       0     .06       0     290     .07       0     360     .06       0
     400     .07       0  525.69     .06       0  535.69      .1       0
   618.1    .045       0  628.78      .1       0  655.69     .06       0
Bank Sta=618.1,628.78
XS Rating Curve= 0 ,0
Exp/Cntr(USF)=0,0
Exp/Cntr=0.3,0.1

Type RM Length L Ch R = 1 ,7386    ,134.8,136.3,137.7
XS GIS Cut Line= 2
 2270632.3730398629774.0772024522271186.05383666630142.663430845
#Sta/Elev= 30
       0 2126.36    56.1 2123.09    94.4 2119.16   117.5 2118.46   142.7 2116.65
   167.9 2117.47     216 2117.74     240 2116.55   267.5  2116.8   279.9  2116.1
   302.1 2117.18   323.2  2117.2   379.4  2116.3     429 2113.71   445.9 2113.74
   457.9 2112.97   501.2 2113.36   510.9 2112.51   542.8  2112.5   558.9 2113.47
   566.8 2112.85   573.6 2109.41   576.4 2108.29   584.8    2108   590.3 2108.38
   591.8 2109.37   595.6 2113.39   600.4 2120.76   604.7 2124.95   665.1 2166.28
#Mann= 6 ,-1,0
       0     .05       0     110     .06       0     120     .05       0
     230     .06       0   573.6    .045       0   591.8     .06       0
Bank Sta=573.6,591.8
XS Rating Curve= 0 ,0
Exp/Cntr(USF)=0,0
Exp/Cntr=0.3,0.1

Type RM Length L Ch R = 1 ,7249    ,99.6,99.6,98.8
XS GIS Cut Line= 2
2270630.39205088629787.286426741 2271079.0843163630249.632951203
#Sta/Elev= 30
       0 2125.95    97.4 2120.08   123.2 2116.54   129.9 2116.14   149.7 2116.17
   203.4 2115.36   220.8 2115.54     261 2114.01     277  2114.6   318.5 2114.22
   324.2 2114.49     404 2114.51   421.8 2113.81   432.6 2112.15   456.3 2112.86
   503.3  2112.7   534.4 2109.56   565.4 2109.82   568.3 2108.79     574 2105.94
   576.8 2105.22   582.5 2105.34  586.26 2105.93   588.4 2106.67     591 2108.74
   594.1  2111.9     599 2115.82   610.2 2123.56   624.9 2132.63   644.3 2143.28
#Mann= 7 ,-1,0
       0     .05       0     270     .06       0     350     .05       0
     410     .06       0     574    .045       0  586.26     .06       0
     620      .1       0
Bank Sta=574,586.26
XS Rating Curve= 0 ,0
Exp/Cntr(USF)=0,0
Exp/Cntr=0.3,0.1

Type RM Length L Ch R = 1 ,7149    ,84.5,86.1,80.4
XS GIS Cut Line= 4
2270588.74994487629917.955011267 2270946.6945223630255.915218186
2270992.73379319  630296.9757372  2271072.695321630320.860349401
#Sta/Elev= 30
       0 2124.49    18.9 2121.87    70.7 2117.92   157.5 2113.58   186.3 2111.18
   219.8 2111.96   268.8 2111.33     296 2112.19   340.3 2111.89   362.3 2111.28
   378.2 2109.98   395.1 2109.37   440.5 2109.38     505 2108.03   508.4 2107.16
   512.92104.694   515.7 2103.75   521.1 2103.53   526.4 2103.71   530.2 2104.64
   533.9 2106.34   542.5  2111.6   547.9 2114.06   553.2 2114.99   561.7  2115.2
   578.4 2113.92     591 2114.52     616 2116.86   624.4 2118.16   637.4 2121.21
#Mann= 8 ,-1,0
       0     .06       0      30     .05       0     170     .06       0
     180     .05       0     320     .06       0   512.9    .045       0
   530.2     .06       0  583.97      .1       0
Bank Sta=512.9,530.2
XS Rating Curve= 0 ,0
Exp/Cntr(USF)=0,0
Exp/Cntr=0.3,0.1

Type RM Length L Ch R = 1 ,7063    ,44.9,44.8,46.1
XS GIS Cut Line= 4
 2270547.5677193629957.9257947872270848.84273468630268.970105933
2270914.48364978630312.7676197112270991.70156256630324.880233481
#Sta/Elev= 30
       0 2125.64    50.8 2120.22    81.4 2117.56     127 2114.94   161.9 2113.65
   182.7 2113.37   196.3  2112.5   216.1 2110.19   294.1 2109.91   317.1 2110.89
   356.3 2110.62   370.5 2109.63   393.1 2109.39   409.1 2107.14   429.9 2107.15
     437 2107.76   446.7 2106.97   467.3 2106.39   473.1 2105.46   481.52102.439
   485.1 2101.66   493.3 2101.52  500.51 2102.44   505.5 2103.88   511.9 2106.83
   514.6  2107.5   529.8 2109.12   538.3 2111.14   554.1 2112.16   590.1 2115.44
#Mann= 6 ,-1,0
       0     .05       0     110     .06       0     380     .07       0
     390     .06       0   481.5    .045       0  500.51     .06       0
Bank Sta=481.5,500.51
XS Rating Curve= 0 ,0
Exp/Cntr(USF)=0,0
Exp/Cntr=0.3,0.1

Type RM Length L Ch R = 1 ,7018    ,102.2,101.1,99.7
XS GIS Cut Line= 4
2270529.23032518629997.1955189842270822.81344424630300.330418726
2270881.42007726630344.9931538772270985.46456339630366.552651003
#Sta/Elev= 30
       0 2124.49    15.7 2122.96    44.5 2119.03      79 2116.53    96.2 2116.06
   116.9  2114.5   149.2 2113.33   178.2 2112.77     194 2111.85   211.2 2110.32
   236.9 2109.68   245.7 2109.07   272.8 2109.11   306.2 2108.27   356.4 2107.77
   400.9 2105.91   420.7 2106.15   449.8 2105.82   453.9 2105.14  462.38 2101.43
   469.6  2100.6   476.2 2100.81   481.12101.439   489.2 2102.26   518.5 2106.47
     523 2107.74     532 2111.61   539.3  2114.2   571.1 2121.59   601.9 2127.89
#Mann= 7 ,-1,0
       0     .05       0     130     .06       0     330     .07       0
     420     .06       0  462.38    .045       0   481.1      .1       0
  535.68     .06       0
Bank Sta=462.38,481.1
XS Rating Curve= 0 ,0
Exp/Cntr=0.3,0.1

Type RM Length L Ch R = 1 ,6917    ,134.6,135.5,136.4
XS GIS Cut Line= 2
2270461.34547802630220.2214812352270947.04149159630493.244941809
#Sta/Elev= 30
       0 2131.43    12.4 2126.29    35.4 2118.15    50.9 2114.23     118 2106.87
   140.8 2105.62   173.4 2105.87   209.7 2104.69   267.2 2105.01   308.8 2104.07
   372.9 2105.19   375.8 2104.77   387.12100.153   392.6 2098.86   397.9 2098.41
   402.5 2098.66   404.92099.913   408.1 2101.99   411.6 2103.35   434.6 2102.53
   439.2 2102.69   443.8 2103.82   450.9 2108.56     461 2119.07   467.2 2124.58
   489.6 2139.44   503.4 2146.41   525.6 2156.01   544.7 2163.97   557.2  2168.3
#Mann= 5 ,-1,0
       0     .05       0     300     .06       0   387.1    .045       0
   404.9     .06       0     410      .1       0
Bank Sta=387.1,404.9
XS Rating Curve= 0 ,0
Exp/Cntr(USF)=0,0
Exp/Cntr=0.3,0.1
